--- MFBgSndyCk.prj (project) ---

Proj Title=MFBgSndyCk
Current Plan=p01
Default Exp/Contr=0,0
English Units
Geom File=g01
Flow File=f01
Plan File=p01
BEGIN DESCRIPTION:
AMEC Environment & Infrastructure, 2013
Projection: NAD 1983 State Plane West Virginia South FIPS 4702 (US Feet)
Vertical Datum: NAVD 1988
END DESCRIPTION:
DSS Export Rating Curves= 0
DSS Export Rating Curve Sorted= 0
DSS Export Volume Flow Curves= 0
DXF OffsetX= 0
DXF OffsetY= 0
DXF ScaleX= 0
DXF ScaleY= 0

--- MFBgSndyCk.p01 (plan) ---

Plan Title=Floodplain
Program Version=4.00
Geom File=g01
Flow File=f01
K Sum by GR=0
Std Step Tol=0.01
Critical Tol=0.01
Num of Std Step Trials=20
Max Error Tol=0.3
Flow Tol Ratio=0.001
Split Flow NTrial=30
Split Flow Tol=0.02
Split Flow Ratio=0.02
Log Output Level=0
Friction Slope Method=1
Unsteady Friction Slope Method=2
Unsteady Bridges Friction Slope Method=1
Global Log Level=0
CheckData=False
Run HTab=0
Run UNet=0
Run PostProcess=0
UNET Theta=0
UNET Theta Warmup=0
UNET ZTol=0
UNET ZSATol=0
UNET MxIter=0
UNET MaxInSteps=0
UNET DtIC=0
UNET DtMin=0
UNET MaxCRTS=0
UNET WFStab=0
UNET SFStab=0
UNET WFX=0
UNET SFX=0
UNET DSS MLevel=0
UNET DZMax Abort=0
UNET Convert EG Bridges=0
UNET Use Existing IB Tables=0
UNET Froude Limit=0
UNET Froude Power=0
Write IC File=0
Echo Input=False
Echo Output=False
Write Detailed=0

--- MFBgSndyCk.f01 (steady flow) ---

Flow Title=NFF Regression Equation
Program Version=4.10
Number of Profiles= 1
Profile Names=P100yr
River Rch & RM=MFBgSndyCk,Main            ,33219.1
922.3438
River Rch & RM=MFBgSndyCk,Main            ,30501.7
974.7829
River Rch & RM=MFBgSndyCk,Main            ,30120.6
1296.954
River Rch & RM=MFBgSndyCk,Main            ,29614.9
1371.412
River Rch & RM=MFBgSndyCk,Main            ,27715.1
1448.743
River Rch & RM=MFBgSndyCk,Main            ,27403.5
1615.266
River Rch & RM=MFBgSndyCk,Main            ,24968.6
 1705.95
River Rch & RM=MFBgSndyCk,Main            ,22023.4
1894.585
River Rch & RM=MFBgSndyCk,Main            ,18123.3
2099.241
River Rch & RM=MFBgSndyCk,Main            ,17656.7
2337.621
River Rch & RM=MFBgSndyCk,Main            ,13930.7
2463.998
River Rch & RM=MFBgSndyCk,Main            ,4296.2
2737.248
River Rch & RM=MFBgSndyCk,Main            ,3522.5
3082.938
River Rch & RM=MFBgSndyCk,Main            ,404.5
3118.366
River Rch & RM=MFBgSndyCk,Main            ,92
6442.896
Boundary for River Rch & Prof#=MFBgSndyCk,Main            , 1
Up Type= 0
Dn Type= 1
Dn Known WS=722.73
DSS Import GetInterval= 0
DSS Import GetPeak= 0
DSS Import FillOption= 0

--- MFBgSndyCk.g01 (geometry) ---

Geom Title=USGS 3m DEM
Program Version=4.10

River Reach=MFBgSndyCk      ,Main
Reach XY= 30
     1937026.358      586482.478     1936743.478      587992.359
     1937016.655      589265.795     1936430.532      590047.901
     1935212.716      590245.619     1933562.728      590971.144
     1932815.565      590761.355     1932092.618      590187.554
     1930410.048      590160.251     1929629.998      588876.903
      1929484.41      589189.617     1928035.977      588867.304
     1927378.276      588983.469     1926012.304      587795.468
     1924863.809      587493.902     1924434.244      586762.993
     1924200.388      585604.986     1923472.299      584837.598
     1922753.002      585395.111        1920939.      584521.034
     1920589.638      583759.251      1920766.77       582963.78
     1920100.609       582063.47     1920376.359      581345.931
      1920218.17      580775.558      1920387.33      580099.753
     1919601.811      580484.354     1919227.915      579832.142
     1918177.538       579904.52     1917325.712      579533.495

Type RM Length L Ch R = 1 ,33219.1 ,206.4,206.2,206
XS GIS Cut Line= 3
     1936469.646      586470.621     1936841.928      586474.872
     1937560.649      586540.223
#Sta/Elev= 30
       0  943.18    19.6  935.02    39.2  928.33    68.6  919.26      98  911.24
   205.8   886.3   264.5  875.19   293.9   871.4   333.1  868.01   401.6  863.92
   479.6  860.76   543.7  855.96   557.6  855.27   568.7  856.16   625.9   869.1
   674.6  881.48   684.4   884.7   694.1  889.12   742.9  915.78   762.4  924.52
   859.9  955.64   889.2  963.45   957.5  979.53   967.2  982.51     977  987.26
  1006.2 1007.79  1025.7 1018.77  1035.5 1022.73  1045.2 1025.42    1094 1035.54
#Mann= 3 , 0 , 0
       0     .06       0   543.7    .045       0   568.7     .06       0
Bank Sta=543.7,568.7
XS Rating Curve= 0 ,0
Exp/Cntr=0.3,0.1

Type RM Length L Ch R = 1 ,33012.8 ,317.1,312,306.9
XS GIS Cut Line= 2
     1936601.619      586661.842     1937277.653      586719.241
#Sta/Elev= 30
       0  915.62    49.2  900.02      59  897.04    68.8  894.35    88.5  889.85
   108.2  885.94   127.8  882.33   157.3  877.43   265.5  860.66   275.3  859.49
   285.2  858.75   344.2  855.22   393.3  851.98   397.1  851.86   403.2  851.66
     413  852.39   422.1  855.18   422.8   855.4   432.6   860.1   442.5  864.44
     472  875.76   481.8  879.93   511.3  894.44     531  903.76   540.8   908.2
   550.6  911.98   580.1   921.1     590  924.28   609.6  930.87   678.5  955.06
#Mann= 3 , 0 , 0
       0     .06       0   397.1    .045       0   422.1     .06       0
Bank Sta=397.1,422.1
XS Rating Curve= 0 ,0
Exp/Cntr=0.3,0.1

Type RM Length L Ch R = 1 ,32700.5 ,206.9,210.4,213.8
XS GIS Cut Line= 3
     1936435.202      587010.521     1936734.753      587032.046
      1937412.78      586963.885
#Sta/Elev= 30
       0  954.18    19.4  950.07    38.8  945.31    96.9  928.71   184.1  904.78
   222.8  895.21   251.9  888.81   300.3  880.67   339.3  873.36   397.7  861.63
   417.1  858.71   436.6  856.99   540.7  849.98   553.4   849.6   565.7  850.37
   572.9  851.32   582.6   853.3     641   867.6   660.5  872.77   670.2  876.36
     680  880.88   728.7  905.23   738.4  909.88   748.1  914.04   816.3   940.1
   923.4  982.66   933.1  987.54   942.8  993.01     972 1010.78   981.8 1016.35
#Mann= 3 , 0 , 0
       0     .06       0   540.7    .045       0   565.7     .06       0
Bank Sta=540.7,565.7
XS Rating Curve= 0 ,0
Exp/Cntr=0.3,0.1

Type RM Length L Ch R = 1 ,32490   ,210.6,215.4,220.2
XS GIS Cut Line= 2
     1936620.752      587203.944     1937264.897      587219.888
#Sta/Elev= 30
       0  897.75    19.5  894.71    29.3  893.48    87.9  887.03   195.3  873.92
   244.1  868.31   253.8  866.61   273.4  862.57   312.4  853.47   322.2  851.67
   331.9  850.77   387.8  847.99   400.3  847.57     410  847.98   412.8   848.4
   419.8  849.44   439.3  853.72   468.6  859.37   478.4  861.74   488.1  864.56
   497.9  867.84   507.7  871.52   517.4  875.52   527.2  879.89     537  884.66
   556.5  894.99   595.5  916.25     615  926.01   624.8  930.26   644.3  937.58
#Mann= 3 , 0 , 0
       0     .06       0   387.8    .045       0   412.8     .06       0
Bank Sta=387.8,412.8
XS Rating Curve= 0 ,0
Exp/Cntr=0.3,0.1

Type RM Length L Ch R = 1 ,32274.7 ,238.7,240.3,241.8
XS GIS Cut Line= 2
     1936517.115      587328.309     1937451.444       587516.45
#Sta/Elev= 30
       0  918.37   117.9  887.94   137.6  883.89     226  868.48   255.5  864.69
   294.8  861.65   373.4  852.22   493.5  846.62   510.9  845.99   518.5   846.8
   520.8  847.04   530.6  850.03   550.2  856.82   589.5  867.73   599.4  870.79
   609.2  874.61     619  879.83   628.8  886.24   697.6  933.22   707.4   939.4
   717.3  944.22   727.1  947.39   756.6  954.95   795.9  966.01     845  980.44
   854.8   983.8   864.6  988.16   923.6 1017.31   933.4  1021.1   953.1 1026.98
#Mann= 3 , 0 , 0
       0     .06       0   493.5    .045       0   518.5     .06       0
Bank Sta=493.5,518.5
XS Rating Curve= 0 ,0
Exp/Cntr=0.3,0.1

Type RM Length L Ch R = 1 ,32034   ,139.3,138.1,137.8
XS GIS Cut Line= 2
     1936579.297       587516.45     1937166.043      587675.892
#Sta/Elev= 30
       0  899.71    68.6  893.41    78.4   892.3    88.3  890.84   107.9  887.51
   127.5  883.91   186.3   872.6   225.6  865.34   235.4  863.34   245.2  860.64
     255  857.11   264.8  852.91   274.6   848.2  278.73  846.67   284.4  844.58
   294.2  843.32     304  843.62   313.8  844.61   362.8  850.07   421.7  856.43
   431.5  857.76   441.3  859.58   470.7  866.19   480.5  868.52   500.2  873.68
     510   876.6   519.8  880.06   529.6  884.53   539.4  889.86     608  928.63
#Mann= 3 , 0 , 0
       0     .08       0  278.73    .045       0     304     .06       0
Bank Sta=278.73,304
XS Rating Curve= 0 ,0
Exp/Cntr=0.3,0.1

Type RM Length L Ch R = 1 ,31896   ,177.1,176.6,175.2
XS GIS Cut Line= 2
     1936518.754      587638.468     1937068.828      587786.749
#Sta/Elev= 30
       0  903.45    78.6  896.28    88.4   895.2    98.2  893.79   117.9  890.22
   186.6  876.93   206.3  873.29   225.9  869.84   235.7  868.23   255.4  865.19
   265.2  863.86     275  861.71   284.8   858.2   294.7  853.75   304.5  848.56
   314.3  844.12   315.9  843.79   324.2  842.05     334  842.15   340.9  842.83
   432.2   852.7   461.7  855.82   471.5  857.39   481.3  859.85   491.1  862.99
     501  866.32   520.6  872.98   550.1  883.14   559.9  886.66   569.7  890.62
#Mann= 3 , 0 , 0
       0     .08       0   315.9    .045       0   340.9     .06       0
Bank Sta=315.9,340.9
XS Rating Curve= 0 ,0
Exp/Cntr=0.3,0.1

Type RM Length L Ch R = 1 ,31719.3 ,320.8,307,293.2
XS GIS Cut Line= 2
     1936274.763      587781.124     1937205.904      587975.643
#Sta/Elev= 30
       0  981.69    98.1  956.65   117.7  951.09   235.4   907.4   245.2  904.24
     255  902.11   264.8   900.9   323.6  896.71   333.4  895.57     353  890.88
   382.5  881.73   402.1  874.98   470.7  850.35   490.3  842.03   493.3  841.22
   500.1  839.39   509.9  838.99   518.3  839.63   617.8   847.8   666.8  853.88
   676.7  855.57   686.5  858.01   774.7  886.77   784.5  888.61   833.6  892.44
   843.4  894.84   853.2  898.66   902.2  921.24   941.4  940.57   951.2  944.58
#Mann= 3 , 0 , 0
       0     .06       0   493.3    .045       0   518.3     .06       0
Bank Sta=493.3,518.3
XS Rating Curve= 0 ,0
Exp/Cntr=0.3,0.1

Type RM Length L Ch R = 1 ,31412.3 ,251.3,250.5,249.8
XS GIS Cut Line= 2
     1936528.276       588256.26     1937086.322      588087.252
#Sta/Elev= 30
       0  901.23    29.2  897.62    38.9  896.24    48.6  894.39    58.3   891.9
      68  888.99   126.3  870.59   213.8  843.61   233.2   836.8   234.7  836.47
     243  834.67   252.7  834.12   259.7   834.3   369.3  839.04   398.4  840.45
   408.2   841.3   417.9  843.23   427.6  846.53   437.3  850.73   476.2  868.68
   495.6   877.4   505.3  881.58     515  884.93   524.8  886.88   534.5  888.15
   544.2  889.04   553.9  889.51   563.6  889.72   573.4  890.43   583.1  892.38
#Mann= 3 , 0 , 0
       0     .06       0   234.7    .045       0   259.7     .06       0
Bank Sta=234.7,259.7
XS Rating Curve= 0 ,0
Exp/Cntr=0.3,0.1

Type RM Length L Ch R = 1 ,31161.6 ,331,330.5,330.1
XS GIS Cut Line= 2
     1936427.828        588559.2     1937343.024       588256.26
#Sta/Elev= 30
       0  919.64    19.7  911.57    29.5  909.09    68.9  901.48   147.6  882.45
   157.4  880.79   206.6  875.86   245.9   872.7   324.6  852.92   383.6  842.48
     417  833.89     423  832.73   432.8  832.26     442   832.7   521.4  836.19
   531.2  837.58     541  840.93   600.1  870.31   619.7  878.36   639.4  883.04
   668.9  887.89   678.8  890.18   688.6  893.03   708.3  900.43   727.9  910.43
   777.1   940.5   796.8  950.05   816.5  956.31   934.5  989.22     964  999.39
#Mann= 3 , 0 , 0
       0     .06       0     417    .045       0     442     .06       0
Bank Sta=417,442
XS Rating Curve= 0 ,0
Exp/Cntr=0.3,0.1

Type RM Length L Ch R = 1 ,30831   ,327.6,329.2,330.8
XS GIS Cut Line= 2
     1936617.563      588830.251     1937223.442      588616.599
#Sta/Elev= 30
       0  905.41    29.2  900.01    38.9  897.61    77.9  885.89   126.5  870.84
     146  865.19     185  854.66   194.7  851.41   214.2  843.83   243.6  831.58
   253.1  829.44   262.8  829.17   268.6  829.47   408.8   836.9   418.6  837.52
   428.3  838.92     438  842.04   447.8     846   467.2  854.43     477  859.03
   506.2  874.04   515.9  878.44   525.6  881.63   535.4  883.62   574.3  889.25
   593.8  892.55   603.5   894.8   613.2  898.32     623  902.73   642.4  912.08
#Mann= 3 , 0 , 0
       0     .06       0   243.6    .045       0   268.6     .06       0
Bank Sta=243.6,268.6
XS Rating Curve= 0 ,0
Exp/Cntr=0.3,0.1

Type RM Length L Ch R = 1 ,30501.7 ,361.9,380.9,399.9
XS GIS Cut Line= 2
     1936509.196      589189.944     1937539.191      588887.005
#Sta/Elev= 30
       0  960.52    97.6  931.76   136.6   920.9     244  899.57   302.6  890.15
   341.6  876.56   361.1  868.47   370.9  863.82   380.6  858.25   400.2  844.86
   409.9  840.11   419.7  836.69   454.3  828.55   458.7  827.67   468.5  827.14
   479.3  827.45   702.7  837.27   712.5   837.8   722.2  839.35     732  843.33
   741.8  849.78     771  871.24   780.8  876.81   790.6  880.25   810.1  883.51
   868.7     891   985.8  913.44  1034.6  925.05  1054.1  928.42  1073.6  930.61
#Mann= 3 , 0 , 0
       0     .06       0   454.3    .045       0   479.3     .06       0
Bank Sta=454.3,479.3
XS Rating Curve= 0 ,0
Exp/Cntr=0.3,0.1

Type RM Length L Ch R = 1 ,30120.6 ,495.3,505.6,516
XS GIS Cut Line= 2
     1936491.604      589209.723     1937550.298      589665.726
#Sta/Elev= 30
       0  964.92    48.8  951.67   136.8  924.41   156.3  919.67   195.4  913.62
   293.1  901.65   332.1  895.12   341.9  892.76     381   881.8   400.5  875.62
   468.9  851.43   478.7  847.25   488.4  841.26   498.2  833.21     508  826.36
  512.61  824.82   517.8  823.12   527.5  822.67   537.3  823.05   752.2  833.53
   810.8  834.18   830.4  835.52     889  843.06   898.7  846.48   947.6  874.02
   957.4  877.92   967.1  880.37   986.6  881.86  1103.9  886.13  1152.7  889.39
#Mann= 3 , 0 , 0
       0     .06       0  512.61    .045       0   537.3     .06       0
Bank Sta=512.61,537.3
XS Rating Curve= 0 ,0
Exp/Cntr=0.3,0.1

Type RM Length L Ch R = 1 ,29614.9 ,441.6,453.7,465.8
XS GIS Cut Line= 2
     1936319.407      589439.319     1937110.239      590226.962
#Sta/Elev= 30
       0 1008.46    29.4  997.23      49  990.61   146.9  964.19   244.8  935.66
   381.8  902.83   440.6  890.47   450.4  886.48   460.2  881.14     470  875.14
   528.7  837.52   548.3   822.6   558.1  818.42   561.8  818.08   567.9  817.53
   586.8  818.37   753.9  828.16   832.2  833.53   861.6  836.16     891  839.68
   920.3  842.01   939.9  844.44   969.3  847.39   988.9  850.72   998.7  853.21
  1018.2  859.68  1057.4   874.1  1067.2  877.19  1086.8   881.6  1116.2  887.43
#Mann= 3 , 0 , 0
       0      .1       0   561.8    .045       0   586.8     .06       0
Bank Sta=561.8,586.8
XS Rating Curve= 0 ,0
Exp/Cntr=0.3,0.1

Type RM Length L Ch R = 1 ,29161.2 ,315.4,323,330.6
XS GIS Cut Line= 2
     1936183.881      589643.405     1936509.143      590536.279
#Sta/Elev= 30
       0  998.48    39.2  983.87    78.4  970.62   127.4  950.16   205.7  926.03
   225.3  921.24   274.3  913.93   284.1  912.26   293.9  909.68   303.7  905.51
   333.1  889.94     431  835.67   440.8  829.76   450.6  822.59   460.4  816.25
   461.4  816.03   470.2  814.06   486.4  814.55   666.2  823.04     676  824.21
   695.6  828.37   734.8  838.81   744.5   841.1   764.1  844.62   773.9  847.93
   813.1  865.85   891.5  905.52   901.3  909.72   911.1  913.02   950.3  923.92
#Mann= 3 , 0 , 0
       0      .1       0   461.4    .045       0   486.4     .06       0
Bank Sta=461.4,486.4
XS Rating Curve= 0 ,0
Exp/Cntr=0.3,0.1

Type RM Length L Ch R = 1 ,28838.1 ,639.9,638.8,637.6
XS GIS Cut Line= 2
     1935990.982      589582.958     1936081.953      590817.924
#Sta/Elev= 30
       0 1044.81      59    1020    88.4 1006.48   137.6  981.19   167.1  963.42
   176.9  960.11   294.8  933.13   383.3  916.15   393.1  913.46   412.8  903.59
   520.9  839.84   530.7  833.07   550.4  816.56   553.8  815.25   560.2  812.77
     570  812.17   578.8  812.37   776.4  817.72   796.1  819.34   815.7  824.53
     855   837.7   884.5  845.69   894.3  850.41   992.6  905.02  1012.3  914.24
  1022.1  916.81  1071.2  923.31  1149.9  937.19    1199  947.28  1238.3  956.91
#Mann= 3 , 0 , 0
       0      .1       0   553.8    .045       0   578.8     .06       0
Bank Sta=553.8,578.8
XS Rating Curve= 0 ,0
Exp/Cntr=0.3,0.1

Type RM Length L Ch R = 1 ,28198.7 ,490.8,483,475.3
XS GIS Cut Line= 2
     1935357.973      589774.147     1935463.204      590733.987
#Sta/Elev= 30
       0  924.85    19.5  923.29    68.3  920.97   146.3   915.7   175.6  914.03
   185.3   913.3   195.1  910.97   204.8  905.89   253.6  874.44   273.1  862.66
   282.8  856.98   292.6  851.68   302.4  847.72   312.1  844.94   351.1  835.26
   429.2  816.42   448.7  810.37   453.1  809.34   458.4  808.09   468.2  807.29
   477.9  807.25   478.1  807.25   653.5  810.18   731.5  812.66   780.3   813.5
   799.8  813.53     829  812.35   848.6  812.36   936.3  816.12   965.6  816.15
#Mann= 3 , 0 , 0
       0     .08       0   453.1    .045       0   478.1     .06       0
Bank Sta=453.1,478.1
XS Rating Curve= 0 ,0
Exp/Cntr=0.3,0.1

Type RM Length L Ch R = 1 ,27715.1 ,313.3,311.3,309.2
XS GIS Cut Line= 2
     1934766.443      589873.001     1935305.357      591148.536
#Sta/Elev= 30
       0  916.62    58.9  903.62    98.2   891.5   117.8  883.46   147.3  865.11
   157.1  861.84     167  861.48   196.4  862.92   225.9  859.68   294.6  842.16
     383  821.65   402.6  818.46   520.5  811.05   595.4  804.41   608.9  803.65
   620.4  803.76   785.6  807.47     874  810.81   913.3  813.91  1031.2  826.13
  1090.1     829  1099.9  830.49  1109.7  834.02  1119.6  839.19  1198.1  882.68
  1266.9  915.12  1286.5  920.82    1316  925.96  1345.4  929.69  1384.7  931.07
#Mann= 3 , 0 , 0
       0     .06       0   595.4    .045       0   620.4     .06       0
Bank Sta=595.4,620.4
XS Rating Curve= 0 ,0
Exp/Cntr=0.3,0.1

Type RM Length L Ch R = 1 ,27403.5 ,385.4,389.7,394
XS GIS Cut Line= 2
     1934471.476      590057.953     1934972.123      591049.682
#Sta/Elev= 30
       0  936.85     9.8  936.98    29.5  935.87   108.1  926.17   157.3  921.86
   206.5  918.64     236   913.3   245.8  910.55   255.6  906.97   265.4  902.79
   285.1  892.73   304.8  881.24   334.3  862.74   353.9  851.19   412.9  818.52
   422.7  813.25   432.6  808.82   442.4  806.25   452.2  805.33   544.7  801.43
   560.4  801.22   569.7  801.36     698  804.06   855.3   808.9     875  810.14
   953.6  824.15     993  830.38  1002.8  833.56  1091.3   868.5  1110.9  877.31
#Mann= 3 , 0 , 0
       0     .06       0   544.7    .045       0   569.7     .06       0
Bank Sta=544.7,569.7
XS Rating Curve= 0 ,0
Exp/Cntr=0.3,0.1

Type RM Length L Ch R = 1 ,27013.9 ,453.6,457.6,461.6
XS GIS Cut Line= 2
     1934211.586      590182.318     1934565.547      591269.711
#Sta/Elev= 30
       0  945.45    39.1  939.78    58.6  935.84   117.3  919.45   175.9  900.48
   205.2  889.87   244.4  873.92   263.9  865.34     303  846.56   322.5  837.98
   342.1   830.6   361.6  824.45   381.2  819.31   400.7  815.34   410.5  814.26
   439.8  813.66   449.6  812.74   459.4  810.72   478.9  803.28   488.7  800.32
   498.5  799.41   508.2  799.52   772.1  808.05   791.7  810.55   860.1   823.8
   879.7  828.62   918.8  839.33   948.1  845.66   957.8  849.34  1143.6  934.31
#Mann= 3 , 0 , 0
       0     .06       0   478.9    .045       0   508.2     .06       0
Bank Sta=478.9,508.2
XS Rating Curve= 0 ,0
Exp/Cntr=0.3,0.1

Type RM Length L Ch R = 1 ,26556.3 ,487.1,492.5,497.9
XS GIS Cut Line= 2
     1933862.408       590287.55     1934047.361      591394.076
#Sta/Elev= 30
       0  972.52    29.5  968.06    78.7  959.02   177.1  939.12   196.8  934.07
   206.7  929.62   216.5  923.84   285.4  878.45     374  822.63   383.8  816.92
   393.6  812.58   423.2   803.9   442.8  799.46   462.5  798.18   526.3   796.6
   541.3  796.36   551.3  796.62   738.1  807.09   767.6  807.75   826.6  807.73
   885.7  810.05   895.5  810.92   925.1  815.31   944.7  816.96   984.1  817.01
  1043.2  818.69    1053  819.96  1072.7  825.85  1082.5  827.68  1121.9  832.23
#Mann= 3 , 0 , 0
       0     .06       0   526.3    .045       0   551.3     .06       0
Bank Sta=526.3,551.3
XS Rating Curve= 0 ,0
Exp/Cntr=0.3,0.1

Type RM Length L Ch R = 1 ,26063.2 ,508.4,517.7,527
XS GIS Cut Line= 2
     1933525.986      590360.893     1933481.342      591448.286
#Sta/Elev= 30
       0  948.84      49   947.7    68.6  945.61    78.4  943.58    88.2  940.68
   107.8  932.87   137.3  916.94   147.1  912.76   225.5  887.93   245.1  878.26
   264.7  869.67   303.9  856.29   392.2  831.24   490.2   814.4   519.6  810.03
   558.9  801.95   578.5  796.79   591.5  794.31   598.1  793.81   616.5  795.26
   637.3   797.5   745.2  796.81     755  798.52   774.6  805.39   813.8  812.52
   882.4  828.87   892.2  831.91     902  836.24   931.4  851.28  1088.3  936.18
#Mann= 3 , 0 , 0
       0     .06       0   591.5    .045       0   616.5     .06       0
Bank Sta=591.5,616.5
XS Rating Curve= 0 ,0
Exp/Cntr=0.3,0.1

Type RM Length L Ch R = 1 ,25545.2 ,572.7,575.9,579.1
XS GIS Cut Line= 2
     1933262.907      590265.228     1932893.002      591196.368
#Sta/Elev= 30
       0  949.33    19.6  942.86    39.3  938.38    58.9   936.2   117.9  932.75
   127.7  931.56   137.5   929.2   225.9   896.7   284.9  878.46   294.7  874.71
   363.4  840.29   402.7  824.05   432.2  814.65   491.1  799.25  507.04  793.98
   520.6  791.22   530.4  791.08  534.91   791.2   726.9  794.17   736.7  795.76
     776  807.06   795.6  810.12   834.9  818.38   854.6  823.63   874.2  830.22
   893.9  837.65   913.5  846.35   933.2   856.6   952.8  868.27  1001.9  900.72
#Mann= 3 , 0 , 0
       0      .1       0  507.04    .045       0  534.91     .06       0
Bank Sta=507.04,534.91
XS Rating Curve= 0 ,0
Exp/Cntr=0.3,0.1

Type RM Length L Ch R = 1 ,24968.6 ,400.8,398.8,396.9
XS GIS Cut Line= 2
     1932875.463      590070.709     1932295.095      591154.913
#Sta/Elev= 30
       0  992.56    78.7  982.59   137.7  974.07   167.2  969.27   186.9  963.93
   196.8  959.33   226.3  942.79   295.1  900.23   334.5  877.75     364  863.52
   413.2  842.69   452.6  824.86   501.7  801.01   521.4  789.66   527.1  787.59
   531.3  786.06   541.1  785.49   552.1  786.23   757.5  799.58     787  802.56
   836.2  809.72   875.6  812.74   944.5  815.78     974  818.74  1003.5  824.57
  1052.7  837.16  1141.2  866.65  1180.6  878.77  1200.2   883.9  1229.8  888.98
#Mann= 3 , 0 , 0
       0      .1       0   527.1    .045       0   552.1     .06       0
Bank Sta=527.1,552.1
XS Rating Curve= 0 ,0
Exp/Cntr=0.3,0.1

Type RM Length L Ch R = 1 ,24569.7 ,673.4,661.8,650.3
XS GIS Cut Line= 2
     1932440.187      590000.554     1932073.471      590816.897
#Sta/Elev= 30
       0  928.16    19.7   917.4    39.3  905.88    49.2  900.99      59  896.72
    98.3  880.78   147.5  859.91   186.8  845.46   216.4  833.76   245.9  821.33
   285.2  804.05   304.9  796.23   324.5  787.33   329.1  786.31   334.4  785.14
     354   784.7   354.1   784.7     413  785.12   511.4  788.48   560.6  791.34
   570.4  792.48   580.2  794.38   609.7  803.25   629.4  806.92   639.2  809.41
   708.1     834   767.1  855.77   816.2  874.44   855.6  891.71   894.9  908.34
#Mann= 3 , 0 , 0
       0     .08       0   329.1    .045       0   354.1     .06       0
Bank Sta=329.1,354.1
XS Rating Curve= 0 ,0
Exp/Cntr=0.3,0.1

Type RM Length L Ch R = 1 ,23907.2 ,646,647.8,649.5
XS GIS Cut Line= 2
     1931721.082      589695.266     1931711.538      590829.652
#Sta/Elev= 30
       0  929.39    29.3  912.26    58.7   896.2    78.2  886.56   107.6  873.45
   127.1  865.99   234.7  828.12   303.2  804.72   342.3   792.7   352.1  790.75
   361.8  790.12   459.6  789.65   537.9  787.51   619.8   784.5   625.9  784.24
   644.8  784.71   684.6  786.21   694.4  786.87   704.1  788.46   733.5  795.61
   782.4  806.34   801.9  809.33   811.7  811.52   821.5  814.78   968.2   869.3
   997.5  881.55  1017.1  890.54  1046.4  905.09    1066  915.34  1134.4  952.26
#Mann= 3 , 0 , 0
       0     .06       0   619.8    .045       0   644.8     .08       0
Bank Sta=619.8,644.8
XS Rating Curve= 0 ,0
Exp/Cntr=0.3,0.1

Type RM Length L Ch R = 1 ,23259.3 ,562.6,567.2,571.9
XS GIS Cut Line= 2
     1931190.163       589793.28     1931129.575      590730.798
#Sta/Elev= 30
       0  972.05    19.6  963.35    39.1  953.56   156.6  888.34   166.4  883.31
   176.2  879.02   225.1  860.84     274  845.73   322.9   831.9   342.5  826.78
   381.7  817.61   391.4  814.61   420.8   803.4   440.4  793.37     460  782.24
     470  779.35   479.5  778.73     495   778.9     548  779.86   616.5  783.18
   655.7  785.67   665.5  786.72   675.2   788.9   714.4   802.1   724.2  804.68
   743.8  808.81   753.5   812.2   890.5  863.77   910.1  872.43   939.5  886.47
#Mann= 3 , 0 , 0
       0      .1       0     470    .045       0     495     .06       0
Bank Sta=470,495
XS Rating Curve= 0 ,0
Exp/Cntr=0.3,0.1

Type RM Length L Ch R = 1 ,22691.8 ,351.4,361.4,371.3
XS GIS Cut Line= 2
     1930710.243      589783.713     1930474.269      590823.274
#Sta/Elev= 30
       0  944.33   107.6  879.11   136.9  863.49   166.3  850.52   195.6  840.33
   215.2  835.79   224.9  835.64   244.5  837.67   264.1  836.84   303.2  831.15
   361.9   820.6   371.6  817.59   381.4  812.24     401  797.72   420.5   780.7
   427.4   777.9   430.3  776.72   440.1  776.45   452.4  777.21   528.1  785.32
   567.2  786.97   616.1  785.26   733.5  787.11   792.2  783.83   831.3  787.53
   899.8  797.74   909.5  797.85   938.9  793.71   968.2  791.77    1066  791.96
#Mann= 3 , 0 , 0
       0      .1       0   427.4    .045       0   452.4     .06       0
Bank Sta=427.4,452.4
XS Rating Curve= 0 ,0
Exp/Cntr=0.3,0.1

Type RM Length L Ch R = 1 ,22330.3 ,292.7,306.5,320.3
XS GIS Cut Line= 2
     1930536.451      589697.615     1929965.649      590555.412
#Sta/Elev= 30
       0  968.04    19.6   961.8    39.2  953.81    98.1  925.26   117.8  914.59
     157  889.84   176.6  880.04   186.4  876.45   225.7   864.6   333.6  833.69
   402.3  815.67   412.1  811.43     422  804.53   431.8  795.67   441.6  785.37
   451.4  777.15     453  776.65   461.2  774.08     471   773.8     478  774.04
   559.3  777.54   569.2   778.8   598.6  789.31   608.4  791.34   677.1  803.68
   726.2  810.24   814.5  826.85   883.2  832.37  1000.9  849.71  1030.4  853.42
#Mann= 3 , 0 , 0
       0      .1       0     453    .045       0     478     .06       0
Bank Sta=453,478
XS Rating Curve= 0 ,0
Exp/Cntr=0.3,0.1

Type RM Length L Ch R = 1 ,22023.4 ,308.7,311,313.2
XS GIS Cut Line= 2
     1930479.052       589656.16      1929442.68      590198.262
#Sta/Elev= 30
       0  960.34   157.3  882.31   186.7  869.17   235.9  850.34   304.7  827.62
   324.3  822.08   383.3  808.04   442.3  786.04   463.7  776.79   471.8   774.2
   481.6  773.46   488.7  773.74   609.4  781.27   619.2  782.09     629  784.47
   638.8  788.94   668.3  804.57     688  813.41   697.8  816.46   776.4   835.9
   825.6  846.24   855.1   856.3   963.2  899.29   982.8  908.58  1051.6  944.45
  1081.1  957.67  1120.4   973.1  1130.3  975.71  1140.1  977.14  1169.6  979.68
#Mann= 3 , 0 , 0
       0      .1       0   463.7    .045       0   488.7     .06       0
Bank Sta=463.7,488.7
XS Rating Curve= 0 ,0
Exp/Cntr=0.3,0.1

Type RM Length L Ch R = 1 ,21711.8 ,312,306.1,300.2
XS GIS Cut Line= 2
     1930335.555       589436.13     1929556.725      589769.408
#Sta/Elev= 30
       0  920.06    97.4   874.6   126.6  860.72   155.8  845.64   165.5  841.68
   175.3  838.78     185  836.88   194.8  835.62   204.5  834.06     224  829.55
   340.8  799.62   360.3  793.52   379.8   786.5   389.5  782.43   399.2  777.94
     409  774.42   413.6  773.76   418.7  773.02   428.4  773.09   438.6  773.57
   486.9  776.75   545.3  781.31   564.8  782.59   574.5  784.36   671.9  809.94
   798.5   843.9   808.2  845.86   827.7  847.98   837.4  849.69   847.1  851.87
#Mann= 3 , 0 , 0
       0      .1       0   413.6    .045       0   438.6     .06       0
Bank Sta=413.6,438.6
XS Rating Curve= 0 ,0
Exp/Cntr=0.3,0.1

Type RM Length L Ch R = 1 ,21405.7 ,1191.8,1174.4,1156.4
XS GIS Cut Line= 2
     1930204.812      589051.875     1929358.176      589654.565
#Sta/Elev= 30
       0  919.75    19.6  909.23    58.8   885.9    68.6  881.08      98  869.59
   127.4  858.83   156.9  848.42   186.3  838.79   225.5  827.18   264.7  814.74
   323.5  799.02   343.2  794.84   362.8  791.84   431.4  785.25   441.2  783.45
   460.8  773.58   470.6  771.32   490.2   772.1   598.1  781.81   627.5  783.66
   647.1  787.37   715.7  806.58   735.3  811.48   745.1  813.45   764.7  816.23
   813.8  826.15   843.2  833.06   911.8  850.41   970.6  869.81  1039.2  894.73
#Mann= 3 , 0 , 0
       0     .08       0   460.8    .045       0   490.2     .06       0
Bank Sta=460.8,490.2
XS Rating Curve= 0 ,0
Exp/Cntr=0.3,0.1

Type RM Length L Ch R = 1 ,20230.5 ,462.9,454.4,445.9
XS GIS Cut Line= 2
      1929491.31      588460.346     1929060.817      589592.383
#Sta/Elev= 30
       0  784.29    68.4  782.84   136.7  780.14   214.9  777.96   234.4  777.88
   263.7  778.41   302.8  777.71   449.3  772.23   654.6  766.86   664.2  766.64
   673.9  767.26   679.6     769   683.7  770.25   693.5  774.92   703.2  779.05
     713  782.57   722.8  785.58   732.5  787.57   752.1  790.44   761.8   792.4
   918.1  825.61     967  835.33   976.7  837.82   986.5  840.73  1025.6  853.08
  1064.6  866.05  1074.4   869.5  1084.2  873.54  1113.5  888.13  1211.1  938.52
#Mann= 3 , 0 , 0
       0     .06       0   654.6    .045       0   679.6     .06       0
Bank Sta=654.6,679.6
XS Rating Curve= 0 ,0
Exp/Cntr=0.3,0.1

Type RM Length L Ch R = 1 ,19775.9 ,474.9,468.4,462
XS GIS Cut Line= 2
     1928842.806      588418.166     1928779.402      589538.173
#Sta/Elev= 30
       0   900.9    68.9  862.88    88.6  852.87    98.4  848.86   127.9  838.73
   177.1  818.38   196.8  812.88   364.1  771.39   383.8  767.73   393.6  767.06
   580.6   765.1   590.4  765.02   600.3   765.6   606.7  767.65   610.1  768.67
   639.6  786.87   659.3  796.59     679  802.13   698.7   809.2   708.5  812.02
   816.8   834.5   846.3  841.14     866  846.37     925  868.44  1003.7   895.6
  1023.4  903.52  1033.2  908.44  1052.9  919.52  1102.1  949.26  1121.8  959.84
#Mann= 3 , 0 , 0
       0     .06       0   580.6    .045       0   606.7     .06       0
Bank Sta=580.6,606.7
XS Rating Curve= 0 ,0
Exp/Cntr=0.3,0.1

Type RM Length L Ch R = 1 ,19307.4 ,716.2,717.4,718.7
XS GIS Cut Line= 2
     1928268.037      588393.558     1928462.113      589525.418
#Sta/Elev= 30
       0  909.86    39.3  890.02    88.3  862.52     108  852.91   176.7  825.84
   245.4   801.9   284.6  793.29   343.5   787.8     422  776.37   480.9  773.22
   490.8   771.7  512.79  765.93     530  764.34   539.8   764.4   579.1  764.82
     638  767.56   647.8  770.11   657.6  774.84   687.1  791.76   696.9  796.24
   726.3   804.8   853.9   832.8   912.8  846.54   952.1  857.44   971.7  864.63
    1011  881.32  1030.6  890.71  1099.3  932.32  1118.9  942.88  1148.4  956.97
#Mann= 3 , 0 , 0
       0     .06       0  512.79    .045       0   539.8     .08       0
Bank Sta=512.79,539.8
XS Rating Curve= 0 ,0
Exp/Cntr=0.3,0.1

Type RM Length L Ch R = 1 ,18589.5 ,437.8,466,494.1
XS GIS Cut Line= 3
     1927630.269      588393.558      1927757.38      589458.452
     1927904.066      589802.846
#Sta/Elev= 30
       0  954.38    49.2  950.31    68.9   946.4   137.8  920.95   186.9  898.64
   216.5  886.48   265.6  869.46   393.6  844.01   482.1   821.6   511.6  809.83
   580.5  768.98   590.3  765.09   600.2  763.02  624.51  759.99   649.4  758.51
  651.91  758.55   747.8  760.64     797  764.51   816.6  767.46   924.9  814.15
  1072.4  849.51  1120.4  864.72  1149.2   876.5  1206.8  903.25  1254.8  923.76
  1293.2  938.93  1341.2  955.67    1370  964.32  1408.4  967.73  1446.8  976.61
#Mann= 3 , 0 , 0
       0     .08       0  624.51    .045       0  651.91     .08       0
Bank Sta=624.51,651.91
XS Rating Curve= 0 ,0
Exp/Cntr=0.3,0.1

Type RM Length L Ch R = 1 ,18123.3 ,470.6,466.4,462.2
XS GIS Cut Line= 4
     1927602.755      588398.665     1927432.775      588789.353
     1926845.837      589257.463     1926303.009      589750.479
#Sta/Elev= 30
       0  953.63    48.4  951.62   106.5   933.6   125.9  924.81     184  891.22
   242.1  868.73     397  830.27   426.1  825.13   494.3  818.49   562.6   790.3
   621.1  757.33   630.8  756.19   647.2  758.76   855.1  761.17   913.6  764.23
   952.6   779.6  1050.1  827.51  1108.6  840.23  1147.6  852.29  1323.5  930.55
  1352.8  941.54  1382.1  945.99  1421.2  948.29  1489.7  947.76  1528.8  942.85
  1538.6  944.46  1597.2     967  1675.5  976.62  1724.3  993.73  1910.1 1033.95
#Mann= 3 , 0 , 0
       0     .08       0   621.1    .045       0   647.2     .06       0
Bank Sta=621.1,647.2
XS Rating Curve= 0 ,0
Exp/Cntr=0.3,0.1

Type RM Length L Ch R = 1 ,17656.7 ,511.5,506.8,502.1
XS GIS Cut Line= 3
     1927352.128      588163.139      1926773.92      588795.355
       1926562.5      588928.813
#Sta/Elev= 30
       0  969.92    19.5  963.03    48.7  949.28   126.6  904.78   155.8  891.21
   175.2  884.22   243.4  863.45   389.4  828.27   457.6  795.47   506.3  774.41
   535.5   757.8   539.3  756.54   545.2  754.59   554.9  754.54   564.3  756.48
   574.4  759.16   584.2  760.12   778.9  762.14   788.6  762.47   798.3  764.62
   808.1  769.91   837.3  790.13   856.8  802.32   914.4  832.98   924.1  837.22
   933.7  840.04   991.4  852.42  1010.6  857.98  1058.7  880.42  1106.8  906.07
#Mann= 3 , 0 , 0
       0     .08       0   539.3    .045       0   564.3     .06       0
Bank Sta=539.3,564.3
XS Rating Curve= 0 ,0
Exp/Cntr=0.3,0.1

Type RM Length L Ch R = 1 ,17149.6 ,837.5,840.7,843.9
XS GIS Cut Line= 3
     1926852.045      587852.126      1926386.33      588579.321
     1926278.465      588792.145
#Sta/Elev= 30
       0  952.32   107.9  902.42   206.1  859.81   215.9  856.45   225.7  854.35
   245.3  851.82     265   847.6   333.6  827.16   372.9   818.8   392.5  810.96
     422  797.53     471  771.18   490.6  762.39   510.3  758.07   544.9  752.76
   559.3  752.11   569.9  752.67   686.9  760.73   706.5     763   716.4  766.15
   765.4  790.25   794.8  803.13   814.5  810.79   853.7   823.7   873.1     827
   930.4  833.11   968.5  840.24  1035.3  849.44  1054.4  855.85  1102.1  880.38
#Mann= 3 , 0 , 0
       0     .08       0   544.9    .045       0   569.9     .06       0
Bank Sta=544.9,569.9
XS Rating Curve= 0 ,0
Exp/Cntr=0.3,0.1

Type RM Length L Ch R = 1 ,16308.8 ,653.5,649.1,644.1
XS GIS Cut Line= 3
     1926389.507      587216.403     1925773.175      587966.167
     1925700.105       588496.72
#Sta/Elev= 30
       0  833.53   127.4  816.55   196.1  805.59   284.3  793.84   333.3  792.31
   421.6   795.1     451  793.75   480.4  787.61   539.2  768.76     549  766.58
   690.4  752.01   705.9  751.26   715.4  751.34   803.9  753.05   813.7  753.41
   823.5  755.22   843.1  764.04   862.7  769.74   911.8  796.91   960.8  819.81
     990  830.59  1009.5  836.32  1077.7  845.59  1145.8  857.18  1272.4  889.05
  1350.3  906.36  1379.6  915.07  1389.3  916.86  1418.5   919.2  1506.1  922.84
#Mann= 3 , 0 , 0
       0     .06       0   690.4    .045       0   715.4     .06       0
Bank Sta=690.4,715.4
XS Rating Curve= 0 ,0
Exp/Cntr=0.3,0.1

Type RM Length L Ch R = 1 ,15658.9 ,591.1,592.8,594.5
XS GIS Cut Line= 3
     1925958.228      586862.901     1925437.906      587464.242
     1925093.304      588131.369
#Sta/Elev= 30
       0  969.99    29.4  968.16    49.1  965.19    88.4  956.68     108  950.24
   127.6  941.33   157.1  923.91   186.5  911.52   225.8  899.61     324  861.72
   392.7  842.78     481  806.48   530.1  787.91   569.4  774.33   618.5   759.8
   638.1  757.01   657.8   756.3     883  754.04   984.2  749.84    1000  749.07
  1009.2  750.47  1029.2  759.04    1078     775  1097.5  783.58    1156  812.57
  1175.5  820.38  1185.3  822.74  1243.8   832.8  1409.6  856.24  1546.1  867.86
#Mann= 3 , 0 , 0
       0     .06       0   984.2    .045       0  1009.2     .08       0
Bank Sta=984.2,1009.2
XS Rating Curve= 0 ,0
Exp/Cntr=0.3,0.1

Type RM Length L Ch R = 1 ,15065.5 ,597.6,612.7,627.7
XS GIS Cut Line= 3
     1925239.445      586704.911     1924708.891      587603.993
      1924463.92      587852.661
#Sta/Elev= 30
       0  887.78    29.3  884.96      78  877.32   175.6   860.8   214.6  855.12
   234.2  851.34   253.7  846.61   292.7  834.98   409.8  796.76   429.3  788.46
   487.8  760.53   497.6  756.66   507.3  754.75   663.4   749.9   835.9  746.08
   848.8     746   860.9  748.16   907.4   764.2   917.1  768.34   985.4  807.76
  1014.7  822.88  1034.2  831.64  1053.6  837.06    1073  840.75  1092.4  843.36
  1140.9  848.34  1160.3  852.62  1199.1  863.87  1247.6  880.17    1393  931.35
#Mann= 3 , 0 , 0
       0     .06       0   835.9    .045       0   860.9     .08       0
Bank Sta=835.9,860.9
XS Rating Curve= 0 ,0
Exp/Cntr=0.3,0.1

Type RM Length L Ch R = 1 ,14452.8 ,508,522,535.9
XS GIS Cut Line= 3
     1925163.198      586561.948     1924299.063      587025.785
     1923968.061      587045.623
#Sta/Elev= 30
       0  852.35    29.4  847.01   117.7  834.35   176.5  829.37   235.4  818.74
   284.4  814.43   313.8  810.06   353.1  801.94   392.3  789.46   470.8   766.3
   490.4  761.97   627.7  748.08   729.4  742.93   745.4  742.41   754.4  743.28
     765  746.34   784.6  754.29     814  764.31   892.5   789.3   912.1   794.2
   941.5  797.04   990.5  816.89    1049  837.88  1107.5  853.11  1117.3  854.34
  1136.8  854.94  1146.6  856.78  1195.3  869.76  1244.1  887.38  1312.4  914.31
#Mann= 3 , 0 , 0
       0     .06       0   729.4    .045       0   754.4     .08       0
Bank Sta=729.4,754.4
XS Rating Curve= 0 ,0
Exp/Cntr=0.3,0.1

Type RM Length L Ch R = 1 ,13930.7 ,363.7,353.5,343.3
XS GIS Cut Line= 3
     1924946.988      586426.802     1924148.059      586416.479
     1923841.931      586497.263
#Sta/Elev= 30
       0  900.42     9.7  898.88    19.5  896.42   107.2  872.32   165.6  857.04
   175.4  853.74   253.3  817.25   360.5  768.86     380  761.18     419  748.94
   428.7  746.88   438.5     746   533.7  742.54   545.7   742.3   555.4  742.64
   558.7   743.5   565.1  745.16   584.6  756.34   613.9  765.76   623.6  769.54
   818.2  849.75   827.8  852.34     847  854.65   866.2  858.11   914.1  868.98
   933.3  874.12   971.7  888.05  1019.7  906.36  1077.2  928.52  1115.6  944.06
#Mann= 3 , 0 , 0
       0     .06       0   533.7    .045       0   558.7     .08       0
Bank Sta=533.7,558.7
XS Rating Curve= 0 ,0
Exp/Cntr=0.3,0.1

Type RM Length L Ch R = 1 ,13577.1 ,371.7,369.9,368.1
XS GIS Cut Line= 3
     1925083.773      585831.245     1924543.689      586009.156
     1923829.996      586272.883
#Sta/Elev= 30
       0  883.44    88.2   856.8   137.3  844.32   147.1  840.22   205.9  807.42
   215.7  802.62   225.5  798.92   245.1  794.17   294.1  787.76     402  777.69
   519.6  761.92   539.2  760.35   597.9  758.93   695.4  750.74   744.2  745.22
   761.9  742.32   773.5  741.61   786.9  742.19     793  742.95   812.5  749.18
   880.8  767.66   890.5  770.49   900.3  774.34  1056.4  851.74  1066.1   855.6
  1075.9  857.72  1124.6  865.27  1173.4   876.3    1232  895.64  1329.5  932.52
#Mann= 3 , 0 , 0
       0     .08       0   761.9    .045       0   786.9     .08       0
Bank Sta=761.9,786.9
XS Rating Curve= 0 ,0
Exp/Cntr=0.3,0.1

Type RM Length L Ch R = 1 ,13207   ,453,442.9,432.7
XS GIS Cut Line= 3
     1924745.311      585532.699     1924013.136      585843.953
      1923704.97      585971.032
#Sta/Elev= 30
       0  933.56    29.5  921.45    88.4  904.34   225.9  859.28   245.6   850.2
   373.2  786.85   422.4  764.47   461.6  748.78   471.5  746.12   481.3  744.88
   530.4  741.74   547.7   741.6  559.88  741.53   572.7  741.79   579.5  742.21
   589.3  744.03   667.9  762.43   687.5  767.96   707.2  774.83   726.8  782.85
   746.5  791.81   766.1  801.78     825   833.6   844.6  843.33   854.4  847.26
   864.2  849.74   913.2  857.84   972.1  870.88  1030.9  891.68  1128.9  924.42
#Mann= 3 , 0 , 0
       0     .06       0   547.7    .045       0   572.7     .08       0
Bank Sta=547.7,572.7
XS Rating Curve= 0 ,0
Exp/Cntr=0.3,0.1

Type RM Length L Ch R = 1 ,12764   ,368,368.5,369
XS GIS Cut Line= 3
     1924683.476      584935.341     1924111.622      585291.161
     1923604.846      585800.933
#Sta/Elev= 30
       0  892.99    97.6  895.09   156.2  892.41   214.7  888.44   312.4  879.11
   429.5  870.51   488.1  856.93   517.3  848.39   546.6  836.21   605.2  807.37
   644.2  792.16   673.5  782.05   731.8  765.89   799.8  744.21   813.4  741.91
   819.2  741.51   838.4  741.75   926.1  750.52   945.5  753.68   955.2  757.35
   984.4  771.74  1071.8  818.03  1110.6  837.29  1130.1  841.68  1217.5  853.55
  1246.6  860.84  1275.8   873.9  1304.9  883.19  1343.8  891.53  1392.3  898.55
#Mann= 3 , 0 , 0
       0     .06       0   813.4    .045       0   838.4     .06       0
Bank Sta=813.4,838.4
XS Rating Curve= 0 ,0
Exp/Cntr=0.3,0.1

Type RM Length L Ch R = 1 ,12395.5 ,528.1,506.1,484
XS GIS Cut Line= 3
     1924110.302      584795.625     1923555.653       585345.17
     1923439.708      585683.093
#Sta/Elev= 30
       0  773.73    58.6  766.28    87.8  763.58   175.7  760.66   312.3  754.69
   439.2  747.65   497.8  742.92     543  740.16   556.3  739.66     568  739.95
   575.8  740.91   585.6  743.74   595.4   747.2   614.9  755.36   634.4  764.58
   673.4  781.96   702.7     794   722.2  800.99   741.8  806.98   751.5  809.47
   761.3  811.35   780.8  813.25   877.4  825.87   896.7  828.01  1022.2  834.23
  1041.5  837.53  1089.8  850.45  1099.4  852.54  1109.1  854.04    1138  856.64
#Mann= 3 , 0 , 0
       0     .06       0     543    .045       0     568     .06       0
Bank Sta=543,568
XS Rating Curve= 0 ,0
Exp/Cntr=0.3,0.1

Type RM Length L Ch R = 1 ,11889.1 ,619.5,601.6,583.8
XS GIS Cut Line= 3
     1923382.123      584244.186     1923401.328      584695.492
     1923408.529      585634.112
#Sta/Elev= 30
       0  895.63    19.6  890.65     108  871.33   137.5  863.49   225.9  831.07
   245.5  822.58     275  807.32   284.8  802.97   314.2  792.25   343.7  783.12
   441.9  760.48     481  754.18   539.7  746.72   565.3  741.45   578.8  739.52
   588.6  739.34   590.3  739.36   950.4   743.2   960.2  744.55   969.9  747.26
   999.3  757.11  1048.2  773.98  1116.6  800.49  1145.9  809.97  1155.7  811.96
  1194.8  816.03  1233.9  816.54  1243.7  817.41  1351.2  839.57  1390.4     845
#Mann= 3 , 0 , 0
       0      .1       0   565.3    .045       0   590.3     .06       0
Bank Sta=565.3,590.3
XS Rating Curve= 0 ,0
Exp/Cntr=0.3,0.1

Type RM Length L Ch R = 1 ,11287.2 ,511.8,529.8,547.8
XS GIS Cut Line= 3
      1922609.26      584736.129     1923192.845      585468.081
     1923399.348      585842.963
#Sta/Elev= 30
       0  874.21    29.2  863.79   136.5  830.61   146.3  829.14     156  829.24
   224.3  832.33   243.8  832.16   302.3  824.94   321.8   821.1   341.3  813.48
   370.6  797.11     390  788.19   438.8  770.29   497.3  752.55   528.2  739.81
   536.3  738.01   553.2  738.53   721.6   741.5   799.6  744.61   819.1  746.96
   916.6  769.75     975  786.18   994.5  792.25  1043.1  811.62    1082  823.61
  1159.8  839.14  1208.5  844.81  1237.7   850.2  1266.8  858.13  1364.1  887.74
#Mann= 3 , 0 , 0
       0      .1       0   528.2    .045       0   553.2     .06       0
Bank Sta=528.2,553.2
XS Rating Curve= 0 ,0
Exp/Cntr=0.3,0.1

Type RM Length L Ch R = 1 ,10757.7 ,743.1,757.5,771.5
XS GIS Cut Line= 3
     1922576.347        584727.4     1922562.274      585882.888
     1922402.693      586150.233
#Sta/Elev= 30
       0  887.67    39.2  873.87    68.6  867.08   166.5  849.86   195.9  846.66
   215.4  843.63   254.6  834.37   293.8  826.64     333  822.23   342.8  820.34
   362.3  813.86   411.3  792.33   430.9   781.7   470.1   757.6   479.9  753.39
   499.4     749   509.2  747.79   538.6  746.08   548.4  744.27     568  739.18
   582.5  736.53   597.4  735.75   607.5  735.94  1067.4  747.05  1155.6  750.39
  1233.4  767.66  1252.9  772.82  1359.9  806.72  1408.6  819.86  1466.9  837.84
#Mann= 3 , 0 , 0
       0     .08       0   582.5    .045       0   607.5     .06       0
Bank Sta=582.5,607.5
XS Rating Curve= 0 ,0
Exp/Cntr=0.3,0.1

Type RM Length L Ch R = 1 ,9998.6  ,513.9,519.1,524.3
XS GIS Cut Line= 3
     1922138.726      584617.644      1921749.74      585422.862
     1921527.437       585578.81
#Sta/Elev= 30
       0  949.87    19.6  940.26    49.1  919.81      59  914.65    68.8  910.62
    78.6  907.54   108.1  901.52   117.9  898.67   167.1  880.73   206.4  864.17
     226  857.08   255.5  847.98   314.5  832.31   383.2  803.76     511  757.36
   530.6  748.65   550.3  738.72   560.1  734.94   569.2   733.5   579.8  733.03
   594.2   733.5   687.9  737.31   884.4  750.15   971.8   762.2   981.5   764.1
   991.2  767.28  1068.8  799.08  1078.5   801.8  1107.6  807.69  1165.8  823.52
#Mann= 3 , 0 , 0
       0      .1       0   569.2    .045       0   594.2     .06       0
Bank Sta=569.2,594.2
XS Rating Curve= 0 ,0
Exp/Cntr=0.3,0.1

Type RM Length L Ch R = 1 ,9479.5  ,554.9,558.2,561.5
XS GIS Cut Line= 3
     1921835.812      584369.243     1921511.546      584801.576
     1921164.467      585263.247
#Sta/Elev= 30
       0  870.51    88.4  850.58   137.6  837.58     167  831.24   186.7  828.18
   206.3  826.29   265.3  824.87     285  822.06   294.8  819.33   334.1  802.71
   353.7  795.68     393  783.09   442.2  769.15     511  735.79   523.6  733.07
   540.4  732.26   548.6  732.38   569.8  733.22   657.9  733.57   667.7  735.02
   677.5   737.6   755.8  762.26   853.7  803.44   873.3  810.99   951.6  827.42
  1010.3  842.28  1039.7  851.39  1069.1  861.57  1088.6  869.57    1118  883.14
#Mann= 3 , 0 , 0
       0      .1       0   523.6    .045       0   548.6     .06       0
Bank Sta=523.6,548.6
XS Rating Curve= 0 ,0
Exp/Cntr=0.3,0.1

Type RM Length L Ch R = 1 ,8920.7  ,505.8,515.3,524.9
XS GIS Cut Line= 3
     1921430.449      584138.601     1920883.824      584709.776
     1920785.338       585167.26
#Sta/Elev= 30
       0  921.18    19.5  912.03    78.1     875    97.6  865.25   185.4  842.28
   234.2  827.74   253.8  819.33   312.3  790.82   341.6  779.57   409.9  757.32
   458.7  736.63   468.5  734.07   478.3  733.52   546.6   732.9   562.1  731.04
   575.9  729.67   587.1     730   634.4  731.56   644.2  732.72     654  735.57
   722.3  763.51   780.8   792.3   800.3  799.47   819.8  804.87   878.3  818.67
   975.8  835.97  1014.8  846.26  1083.1  866.73  1161.1  880.94  1258.6  901.46
#Mann= 3 , 0 , 0
       0     .06       0   562.1    .045       0   587.1     .06       0
Bank Sta=562.1,587.1
XS Rating Curve= 0 ,0
Exp/Cntr=0.3,0.1

Type RM Length L Ch R = 1 ,8405    ,421.1,431.3,441.4
XS GIS Cut Line= 3
      1921301.58      583877.987     1920321.404      584371.416
     1920041.989      584404.145
#Sta/Elev= 30
       0  872.65    39.2  870.85      98  865.16   137.2  857.78   186.2  851.04
   225.4  841.88   274.3  832.58   323.3  815.75   450.7  765.08   499.7  737.25
   509.5  733.41   519.3  731.84   578.1  729.41   597.7  728.14   607.5  729.22
   627.1  733.43   744.6  735.04   813.2  740.46   901.4  767.63   960.2  783.41
   999.4  798.35    1019  804.38  1107.1  821.05  1136.2  822.74  1194.4  819.35
  1242.9  819.45  1262.3  820.48  1291.4  826.87  1310.8  829.41  1378.7  828.64
#Mann= 3 , 0 , 0
       0     .06       0   578.1    .045       0   607.5     .06       0
Bank Sta=578.1,607.5
XS Rating Curve= 0 ,0
Exp/Cntr=0.3,0.1

Type RM Length L Ch R = 1 ,7973.5  ,845.8,842.2,838.5
XS GIS Cut Line= 3
     1921363.546      583702.678     1920181.146      583814.388
     1919441.336      583669.827
#Sta/Elev= 30
       0  842.46    78.5  833.23   137.4  831.95   186.5  835.94   215.9   834.5
   274.8  822.34   431.9  773.97   569.3  741.42   598.7  737.66   716.5  733.61
   765.6  727.67   785.2  725.77     795  726.44   834.3   730.8   893.2   731.7
  1030.6   742.5  1050.2  745.76  1109.1  763.77  1226.8  828.18  1285.6  837.57
  1373.7  855.17  1471.6  881.78  1579.2  892.56  1657.6  902.84  1716.3  921.74
    1775  949.32  1794.6  956.45  1843.6  966.13  1902.3  969.23  1941.5  976.49
#Mann= 3 , 0 , 0
       0     .06       0   765.6    .045       0     795     .06       0
Bank Sta=765.6,795
XS Rating Curve= 0 ,0
Exp/Cntr=0.3,0.1

Type RM Length L Ch R = 1 ,7130.9  ,739.7,724.4,709
XS GIS Cut Line= 3
     1921582.756      582784.535     1920568.662        583027.1
     1920147.961       583062.99
#Sta/Elev= 30
       0  951.42    19.7  935.94    29.5  930.39    88.5  907.21   137.7  889.17
   245.9  851.53   295.1  839.32   314.8  835.05   344.3  830.21   354.1  827.22
   383.6  812.36   403.3  803.43   452.5   783.1   501.7  764.27   511.5  761.65
   521.4  760.23   737.8  735.86   806.6   729.4     823   726.3   836.1  724.62
     848  725.58   895.2  735.39   934.5  746.93  1013.2  774.27  1121.2  816.46
  1170.4  833.63  1229.3  849.27  1307.8  872.57  1386.4  893.65  1464.9  911.63
#Mann= 3 , 0 , 0
       0     .06       0     823    .045       0     848     .08       0
Bank Sta=823,848
XS Rating Curve= 0 ,0
Exp/Cntr=0.3,0.1

Type RM Length L Ch R = 1 ,6406.1  ,541.9,560.3,578.6
XS GIS Cut Line= 3
     1920797.709      582073.747     1920444.795      582335.904
     1919955.094      582808.758
#Sta/Elev= 30
       0  928.35     9.8  925.66   107.5   893.3   234.5  860.45     254  854.29
   332.2  820.95   351.7  811.12     381  794.95   400.6  785.99   420.1  779.78
     498  757.22   556.3  735.85   575.8  727.17   583.9  724.22   585.5  723.64
   595.2  723.08   608.9  725.14   614.7  726.44   624.4  727.39   682.8     730
   692.5  732.07   702.2  735.81   731.4  751.56   741.1  756.09     780  771.58
   925.9  832.51   935.6  836.12   945.3  838.82  1013.4  852.89  1120.4   866.7
#Mann= 3 , 0 , 0
       0     .08       0   583.9    .045       0   608.9     .06       0
Bank Sta=583.9,608.9
XS Rating Curve= 0 ,0
Exp/Cntr=0.3,0.1
